HEC-RAS study HLLSCK.prj: HLLSCK

--- HLLSCK.g01 (geometry) --- (continued)

Type RM Length L Ch R = 1 ,32357   ,228.7,245.8,255.5
XS GIS Cut Line= 2
2159368.23797985428965.877098389 2159055.6483051428934.031501498
#Sta/Elev= 30
       0 3404.25    12.1 3400.49    32.2 3391.69    44.3 3384.09    56.4 3375.43
    64.4 3368.51    73.7 3359.54    88.5 3342.83   108.6 3321.82   116.7 3308.29
   124.7 3299.37   128.7 3292.26   132.7 3287.07   139.4 3285.68   146.7 3284.93
   164.9 3284.75   169.4 3285.31     173 3285.85     181  3285.7   186.8 3287.17
   197.1 3291.98   213.2 3296.26   223.3 3301.72   237.3  3310.6   261.4 3327.21
   273.5 3334.24   281.3 3344.98   285.5 3349.47   292.6 3355.92   314.2 3370.98
#Mann= 5 ,-1,0
       0      .1       0   139.4    .045       0   169.4      .1       0
     170     .06       0     270      .1       0
Bank Sta=139.4,169.4
XS Rating Curve= 0 ,0
Exp/Cntr(USF)=0,0
Exp/Cntr=0.3,0.1

Type RM Length L Ch R = 1 ,32111   ,311.4,310.3,304.2
XS GIS Cut Line= 2
2159422.33824825428835.2356585132159196.06690192428636.899046298
#Sta/Elev= 30
       0 3353.32     9.2 3343.82      20 3335.27    28.5 3326.95    45.4 3312.19
      72 3292.64    76.7 3289.94      82 3285.33      88 3281.46    94.1 3278.63
     105 3276.26   109.3 3276.14   118.4 3277.92   124.9 3278.39   133.4 3276.79
   142.7 3275.04   170.2 3276.39   175.9  3276.4   181.6 3277.34   197.3  3284.7
   209.4  3292.4   215.6 3293.96     221 3296.85   231.6 3306.04   243.9 3314.97
   258.1 3323.67   270.1 3333.87   282.3 3342.69   289.3 3349.47   300.9 3363.33
#Mann= 4 ,-1,0
       0      .1       0   133.4    .045       0   170.2     .06       0
     280      .1       0
#XS Ineff= 2 , 0
          122.75  3294.8
Permanent Ineff=
       F       F
Bank Sta=133.4,170.2
XS Rating Curve= 0 ,0
Exp/Cntr(USF)=0,0
Exp/Cntr=0.3,0.1

Type RM Length L Ch R = 1 ,31801   ,219,213.8,201.5
XS GIS Cut Line= 2
2159671.93123637428646.3427447292159362.18839038428424.574198191
#Sta/Elev= 30
       0 3359.85     8.9 3354.53    15.7 3349.66    24.3 3343.26    46.5 3325.33
    72.3 3306.33    86.7  3291.8    95.3 3281.02     101 3272.18     103 3269.85
   106.7 3267.62   132.5 3267.03   149.7 3267.39     160 3268.89   178.4 3270.58
   186.6 3270.31   201.3 3268.72   211.2 3269.28     226 3268.28   240.8 3269.93
   256.2 3270.03   281.6 3269.33   294.9  3266.8   304.7 3268.38   309.6 3268.47
   314.6 3270.11   319.5 3273.03   331.8 3282.49   345.6 3290.74   380.9 3323.94
#Mann= 5 ,-1,0
       0      .1       0   106.7    .045       0   149.7      .1       0
     160     .06       0     330      .1       0
#XS Ineff= 2 , 0
                          179.71         3302.46
Permanent Ineff=
       F       F
Bank Sta=106.7,149.7
XS Rating Curve= 0 ,0
Exp/Cntr(USF)=0,0
Exp/Cntr=0.3,0.1

Type RM Length L Ch R = 1 ,31587   ,102.8,94.1,87.3
XS GIS Cut Line= 3
2159729.24966504428513.8771931362159592.52866668428425.671535599
2159442.81534223428317.063591726
#Sta/Elev= 30
       0 3322.33    20.3 3307.69    38.2 3296.84    44.1 3294.21    56.3 3289.84
    82.3 3276.42    97.2 3270.24   104.6 3268.55   115.5 3268.14   141.5 3268.68
   160.4 3270.68   168.1 3270.68   183.4 3268.04   192.8 3265.79   202.7 3264.32
   209.1 3262.12     212 3261.31   214.9 3261.16   232.3 3261.67   252.1 3261.81
   265.7 3264.62   276.8 3266.04   279.3 3267.07   286.5 3271.25   299.8 3282.45
   311.4 3291.13   326.2 3301.04   331.2 3303.22   340.7 3309.46   347.7 3315.91
#Mann= 3 ,-1,0
       0      .1       0   209.1    .045       0   232.3      .1       0
Bank Sta=209.1,232.3
XS Rating Curve= 0 ,0
Exp/Cntr(USF)=0,0
Exp/Cntr=0.3,0.1

Type RM Length L Ch R = 1 ,31493   ,187.1,195.6,203.1
XS GIS Cut Line= 3
2159698.25376759428298.1239228692159635.90198285428308.515886992
2159468.64084602428296.144501131
#Sta/Elev= 30
       0 3282.94    10.2 3279.82    22.4 3277.18      71 3268.25      75 3265.11
      79 3254.84      83 3243.53      87  3237.2      95 3231.68    99.7 3227.35
   103.4 3223.24   106.9 3218.55   111.1 3216.07   119.1 3215.76   125.8 3216.14
   135.1 3214.03   139.1 3213.89   143.2  3214.2   147.2 3215.25   151.2 3217.18
   155.2 3218.43   159.4  3221.2   171.2 3231.12   179.3  3234.8   183.3  3237.2
   191.3  3244.7   199.3 3250.76   207.3 3263.32   222.9 3281.05   230.9 3289.11
#Mann= 3 ,-1,0
       0      .1       0   111.1    .045       0   125.8      .1       0
Bank Sta=111.1,125.8
XS Rating Curve= 0 ,0
Exp/Cntr(USF)=0,0
Exp/Cntr=0.3,0.1

Type RM Length L Ch R = 1 ,31297   ,94.4,94.7,95.2
XS GIS Cut Line= 2
2159740.42044933428209.9288667132159579.54152209 428078.23894315
#Sta/Elev= 30
       0 3282.42     1.2  3281.2     5.5  3275.2    20.1 3254.02    23.4 3250.44
    31.3 3243.29      49  3229.4    57.2 3221.86    70.6 3211.51    83.1  3203.9
    93.4 3198.78    97.4  3197.4   103.7 3193.85   108.5 3192.93     114 3193.46
   121.2 3193.32   124.4 3193.86   139.9 3194.18   142.8 3195.46   145.1 3196.93
   160.6 3212.23   165.6 3218.24   168.4 3225.17   171.7 3234.25   174.1 3239.36
   176.9 3244.73   184.3 3256.71   191.6 3270.29   196.7 3276.58   207.9 3281.48
#Mann= 3 ,-1,0
       0      .1       0   103.7    .045       0   124.4      .1       0
Bank Sta=103.7,124.4
XS Rating Curve= 0 ,0
Exp/Cntr(USF)=0,0
Exp/Cntr=0.3,0.1

Type RM Length L Ch R = 1 ,31203   ,164.5,157.9,152.8
XS GIS Cut Line= 2
2159807.81576027428146.908401508 2159599.8260537427967.900867169
#Sta/Elev= 30
       0 3284.25     4.8 3281.84     6.6 3280.03    14.9  3269.2    20.6 3263.41
    26.5 3254.15    31.2 3244.27      35 3240.29    45.6  3234.8    51.7 3230.51
    60.5 3222.52    68.1 3217.77    74.7 3211.95      84 3207.52   100.2  3193.4
   110.4 3188.12   119.2 3187.08   125.8 3187.97   137.6 3187.83   143.7 3188.73
   168.4 3201.85   189.5 3214.69   210.9 3231.66   217.3 3240.41   223.4 3251.72
   229.5  3264.5   236.4 3270.09   247.7 3277.92   260.2 3281.16   274.4 3282.91
#Mann= 3 ,-1,0
       0      .1       0   110.4    .045       0   125.8      .1       0
Bank Sta=110.4,125.8
XS Rating Curve= 0 ,0
Exp/Cntr(USF)=0,0
Exp/Cntr=0.3,0.1

Type RM Length L Ch R = 1 ,31045   ,137.6,142,145.8
XS GIS Cut Line= 4
2159862.30198722427966.2929801922159839.75857299427938.801011613
2159757.28266725427921.2061517232159674.80676151427925.604866695
#Sta/Elev= 30
       0 3219.76     5.1 3214.67    19.4 3202.83    27.9 3196.31    34.9 3192.69
    39.2 3188.88    43.3  3184.5    47.4 3181.53    62.5 3173.87    71.9 3168.33
      76 3168.93    83.8 3168.64    88.3 3167.41    92.4 3168.58    95.3 3168.84
   100.8 3169.35   107.4 3169.17   112.8 3170.03     129 3176.39     137 3181.25
     149 3187.62     157  3193.5   161.1 3195.96   165.1  3200.2   170.3 3209.99
   173.1  3214.1   181.1 3221.91   189.4 3226.77   197.2 3232.44   202.5 3235.46
#Mann= 3 ,-1,0
       0      .1       0    83.8    .045       0    95.3      .1       0
Bank Sta=83.8,95.3
XS Rating Curve= 0 ,0
Exp/Cntr(USF)=0,0
Exp/Cntr=0.3,0.1

Type RM Length L Ch R = 1 ,30903   ,176.1,175.2,171.6
XS GIS Cut Line= 3
2159905.88821764427868.1744334582159879.07087289427822.920164193
2159775.99170401427755.876802317
#Sta/Elev= 30
       0 3150.86     3.5 3148.56     8.1 3145.05    19.1 3137.87    22.1 3135.51
    31.4 3128.88    40.7 3120.83    45.3 3117.36    53.1 3110.58    64.6 3101.39
    67.5 3099.61    76.2 3096.41    79.9 3095.23    84.7 3094.82    87.8  3095.4
    89.5 3095.45    92.5 3096.38      99 3099.37   103.8 3101.25   113.3 3106.84
   118.1 3109.35   122.5 3112.12   128.2 3115.99   137.2 3121.51   145.6    3128
   151.5 3132.77   156.3 3136.31     161 3140.23   170.6 3146.88   175.6  3150.7
#Mann= 3 ,-1,0
       0      .1       0    76.2    .045       0    92.5      .1       0
Bank Sta=76.2,92.5
XS Rating Curve= 0 ,0
Exp/Cntr(USF)=0,0
Exp/Cntr=0.3,0.1

Type RM Length L Ch R = 1 ,30728   ,273.8,276.2,275.3
XS GIS Cut Line= 2
2160018.85176073427700.7471510982159845.37706188427618.535228598
#Sta/Elev= 30
       0 3130.64    11.8 3122.26    17.7 3117.78    25.1 3112.44    34.7 3105.98
    42.8 3101.29    64.4 3086.32    67.8 3084.39    70.8  3082.1    73.8  3079.4
    76.8 3078.12    78.2  3076.9    83.1 3073.79    87.1 3073.29    91.5 3073.28
   100.3 3073.07   109.2 3073.31   118.1 3074.39   122.5 3075.71   126.9 3077.97
   131.3 3081.41   136.8 3086.74   139.8 3089.44   144.6  3093.3   153.5 3099.06
   157.9 3102.54   166.7 3109.94     180 3120.76   188.9 3127.17     192 3129.16
#Mann= 3 ,-1,0
       0      .1       0    91.5    .045       0   109.2      .1       0
Bank Sta=91.5,109.2
XS Rating Curve= 0 ,0
Exp/Cntr(USF)=0,0
Exp/Cntr=0.3,0.1

Type RM Length L Ch R = 1 ,30452   ,208.8,201.7,194.9
XS GIS Cut Line= 3
2160085.97892681427480.5097073382160061.08907871427431.484248967
2159937.39407605427359.077418141
#Sta/Elev= 30
       0 3078.72       4 3077.13     8.2 3074.31    12.7 3070.61    17.2 3068.01
    21.7    3066    30.6 3061.03    45.5 3054.53    53.1 3051.81      56 3050.35
    60.7 3047.41    65.3 3045.07    79.2 3040.16    88.5 3035.64    92.4 3034.63
    99.1  3033.3   102.4 3033.53   105.5 3034.82   107.1 3035.58     110 3038.07
   120.9 3048.76   124.6 3051.38   134.8 3057.68   139.5 3059.85   148.7 3061.39
   153.8 3063.11   162.5 3068.08   168.4 3070.59   181.2 3077.27   198.3 3083.93
#Mann= 3 ,-1,0
       0      .1       0    92.4    .045       0   105.5      .1       0
Bank Sta=92.4,105.5
XS Rating Curve= 0 ,0
Exp/Cntr(USF)=0,0
Exp/Cntr=0.3,0.1

Type RM Length L Ch R = 1 ,30250   ,213.9,226,238
XS GIS Cut Line= 3
2160268.52726644427270.0006209522160201.32467658427236.399326022
2159958.17348781427232.122797576
#Sta/Elev= 30
       0 3057.18     6.8 3054.83    24.7 3050.19    63.5 3042.81    89.3  3036.8
   108.3 3033.72   116.3 3033.02   120.3 3031.89   124.3 3029.82   128.3 3026.14
   136.3  3016.3   140.3 3012.05   144.3 3009.02   150.2 3006.98   152.3 3006.41
   168.3 3006.75   185.6 3007.98   192.3 3007.56   196.3 3006.66   208.3 3007.02
   212.3 3007.77   216.3  3009.3   232.3 3018.17   236.7 3020.05   244.1 3025.33
   256.3 3035.88   264.4  3041.4   296.3 3058.62   312.3 3066.68   318.3 3070.73
#Mann= 3 ,-1,0
       0      .1       0   150.2    .045       0   168.3      .1       0
Bank Sta=150.2,168.3
XS Rating Curve= 0 ,0
Exp/Cntr(USF)=0,0
Exp/Cntr=0.3,0.1

Type RM Length L Ch R = 1 ,30024   ,321.5,289.5,278.3
XS GIS Cut Line= 3
2160255.65944053427220.0015335072160200.50957106427090.657289567
2160117.54341073427005.428415784
#Sta/Elev= 30
       0 3046.35      17 3043.17    29.3 3041.83    46.6 3038.14    68.3 3030.54
    81.3 3023.55    90.2 3020.53   100.7  3017.8   116.1 3011.77   126.7 3008.82
   137.9 3004.79   147.6 3000.41   152.6 2997.33   158.9 2992.62   167.4 2984.48
   170.2 2981.51   175.5 2977.75   184.3 2977.58   204.1 2977.03   209.8 2977.03
   212.6 2977.43   215.6 2977.91   221.4 2980.03   223.9 2983.11   232.8 2995.87
   235.2  2998.6   238.6 3002.16   249.4 3011.63     255 3017.86   259.6 3021.14
#Mann= 3 ,-1,0
       0      .1       0   184.3    .045       0   212.6      .1       0
Bank Sta=184.3,212.6
XS Rating Curve= 0 ,0
Exp/Cntr(USF)=0,0
Exp/Cntr=0.3,0.1

Type RM Length L Ch R = 1 ,29734   ,398.9,431.4,451.4
XS GIS Cut Line= 3
2160486.38406436426816.0536713312160304.84853849426863.161843244
2160215.46629999426907.891303711
#Sta/Elev= 30
       0 3013.49     7.1 3012.61    22.9 3011.65    31.2 3010.47    39.5 3010.16
    47.7 3009.21      52 3008.02      56 3004.88    61.8 2998.03    68.4 2989.92
    72.5 2983.74    76.7  2976.7    84.8 2969.08    89.1 2964.11    93.2 2958.02
    97.3 2953.29   113.9 2939.93     118 2938.65   131.9 2937.19   151.1 2938.55
   163.4 2938.38   192.5 2947.66   201.7 2949.52   218.9 2956.27   224.1 2957.72
     233 2962.38   255.4 2970.57   268.8 2974.66     282 2977.74   287.5 2979.63
#Mann= 3 ,-1,0
       0      .1       0     118    .045       0   151.1      .1       0
Bank Sta=118,151.1
XS Rating Curve= 0 ,0
Exp/Cntr(USF)=0,0
Exp/Cntr=0.3,0.1

Type RM Length L Ch R = 1 ,29303   ,463.5,454.5,438.1
XS GIS Cut Line= 2
2160563.01950652426747.5119723552160387.03479737 426452.31181507
#Sta/Elev= 30
       0 3004.32    21.3 2995.82    36.8 2988.21    52.4 2982.07    75.9 2968.66
    86.5  2961.2    91.2 2957.17    94.2 2952.14   100.5 2943.32     103 2941.08
   111.7  2933.7   120.5 2927.24   133.1 2916.42   137.8 2913.75   155.5 2912.22
   170.1  2913.7   185.2 2911.95   200.8 2911.52   208.7 2911.89   216.9 2912.65
   219.7 2914.47   221.6  2916.1   235.6 2931.95   251.8 2936.79   272.2    2941
   286.8 2946.53   307.2 2957.41     316  2960.9     338 2974.81   343.7 2977.63
#Mann= 3 ,-1,0
       0      .1       0   185.2    .045       0   208.7      .1       0
Bank Sta=185.2,208.7
XS Rating Curve= 0 ,0
Exp/Cntr(USF)=0,0
Exp/Cntr=0.3,0.1

Type RM Length L Ch R = 1 ,28849   ,416.2,412.9,406.8
XS GIS Cut Line= 3
2161061.16977194426507.6618445612160997.30435329426382.769470325
2160619.78876753426255.038633038
#Sta/Elev= 30
       0 2956.04    14.5 2948.19    23.4 2942.16    29.7 2937.44    47.7 2921.81
    52.2 2918.82    59.1 2916.12    76.9 2911.69   110.6 2908.25   140.3 2903.42
   199.2 2901.58   255.5 2896.94   276.6 2897.51   284.4 2895.47   297.7 2889.16
   301.9 2888.52   318.8 2888.83   343.8 2888.88   352.6 2889.12     361 2892.78
   365.3 2893.39   391.7 2893.97   399.1 2897.86   415.9 2910.82   424.4    2916
   437.1 2920.49   479.3 2938.33   487.7 2940.77   508.8 2951.23   538.8 2962.76
#Mann= 3 ,-1,0
       0      .1       0   318.8    .045       0   343.8      .1       0
Bank Sta=318.8,343.8
XS Rating Curve= 0 ,0
Exp/Cntr(USF)=0,0
Exp/Cntr=0.3,0.1

Type RM Length L Ch R = 1 ,28436   ,224.4,234.8,245.2
XS GIS Cut Line= 2
2161160.93777432425929.0076577882160713.75211298425906.016107076
#Sta/Elev= 30
       0 2928.69    16.8 2916.54    48.8  2896.9    56.8  2893.1    84.9 2882.36
    92.9 2880.15   104.9 2879.24   116.9 2879.34   136.9 2874.43     153  2875.4
     169 2871.55     193 2872.53   221.1 2872.32   232.9 2870.84   241.1 2872.39
   273.1 2871.43   293.9 2872.68   305.2 2873.97   309.2 2873.13   312.9 2871.12
   317.7 2869.98   337.2 2870.22     343 2871.16   353.2 2874.56   372.6 2884.54
   385.3 2893.39   397.3 2903.35   421.3 2919.22   441.3 2928.75   447.8 2930.73
#Mann= 3 ,-1,0
       0      .1       0   312.9    .045       0     343      .1       0
#XS Ineff= 2 , 0
           240.1 2892.67
Permanent Ineff=
       F       F
Bank Sta=312.9,343
XS Rating Curve= 0 ,0
Exp/Cntr(USF)=0,0
Exp/Cntr=0.3,0.1

Type RM Length L Ch R = 1 ,28201   ,243,248.9,272.3
XS GIS Cut Line= 3
2161176.43704636425901.5454192282161109.78717075 425836.06483968
2160794.07723364425624.422252213
#Sta/Elev= 30
       0 2931.46      40 2911.29    63.3 2901.31    90.1 2884.68   100.2 2879.29
   109.8 2876.03   129.1 2873.16   153.2 2871.72   172.4 2871.63   180.3 2868.77
   188.9 2864.13   196.5 2862.75   215.8 2863.78   230.2 2866.12   273.6 2862.85
   302.4 2865.18     310 2864.93   327.3 2862.45   342.9 2862.45   360.2  2862.3
   367.7 2862.51   379.5 2862.64     386 2864.18   400.3 2875.35   407.5 2882.08
   410.9 2886.23   416.7 2891.91   425.3 2897.26   442.1 2901.06   473.5 2905.41
#Mann= 3 ,-1,0
       0      .1       0   342.9    .045       0   367.7      .1       0
#XS Ineff= 2 , 0
          303.38 2879.68
Permanent Ineff=
       F       F
Bank Sta=342.9,367.7
XS Rating Curve= 0 ,0
Exp/Cntr(USF)=0,0
Exp/Cntr=0.3,0.1

Type RM Length L Ch R = 1 ,27952   ,341.5,342.5,341.1
XS GIS Cut Line= 4
2161164.38650693425818.6482143722161105.75805262425748.523984701
2161025.28762513425407.0994566342161022.98847005425334.676071892
#Sta/Elev= 30
       0 2901.44    15.4 2894.78    62.7 2877.89    69.3 2876.34    81.4 2875.24
    99.1 2866.93   112.1  2862.9   201.7 2857.37   225.2 2853.53   246.9  2854.6
   259.2 2854.05   275.7 2855.83   298.4 2853.68   320.9 2853.19     325 2852.75
   337.3 2849.19   349.6 2848.06     368 2849.46   386.6 2849.24   401.5 2850.66
   407.2 2853.34   411.4 2857.39   415.4 2860.14   429.6 2860.24   435.9 2861.33
     440 2863.61   480.1 2893.07   492.1 2900.55   496.1 2902.35   514.6  2904.9
#Mann= 4 ,-1,0
       0      .1       0   337.3    .045       0     368     .06       0
  452.18      .1       0
Bank Sta=337.3,368
XS Rating Curve= 0 ,0
Exp/Cntr(USF)=0,0
Exp/Cntr=0.3,0.1

Type RM Length L Ch R = 1 ,27610   ,354.7,356.1,354.4
XS GIS Cut Line= 2
2161439.30882435425706.2808211682161342.74431136 425284.38586561
#Sta/Elev= 30
       0 2889.71    10.2 2885.06    30.2 2874.06    54.5 2863.29    62.7 2860.45
   103.7 2849.13   111.9 2848.85   128.3    2850   163.8 2847.28   173.5 2845.19
   185.8 2840.62   198.1 2839.45   214.5 2839.56   260.7  2842.1   280.2 2839.44
   288.4 2836.42   297.4 2835.79   308.9 2834.97   321.2 2835.06   327.2 2835.77
   337.6 2839.53   341.7  2840.4   358.1 2840.66   362.2 2841.63   366.3  2843.8
   370.4 2845.07   399.2 2847.07   403.3 2848.07   423.8 2862.76   432.8 2870.08
#Mann= 4 ,-1,0
       0      .1       0   297.4    .045       0   327.2     .06       0
     410      .1       0
Bank Sta=297.4,327.2
XS Rating Curve= 0 ,0
Exp/Cntr(USF)=0,0
Exp/Cntr=0.3,0.1

Type RM Length L Ch R = 1 ,27253   ,369.4,350.2,317.5
XS GIS Cut Line= 3
2161776.13504228425621.2120835352161676.12179668425301.629528643
2161556.56573298425252.197694613
#Sta/Elev= 30
       0 2917.78    22.3  2895.9    46.1 2875.77    63.8 2859.08      83 2842.66
    92.2 2836.15    96.4 2834.01     109 2829.45   118.1 2827.35   125.8 2823.84
   137.3 2822.27   146.7 2822.28   163.5 2825.76   178.8 2826.97   192.8 2824.63
   220.3 2822.46   230.6 2822.05   244.1 2822.36     249 2823.24   255.7 2827.44
   259.9 2829.21   289.2 2833.45   310.2 2832.56   331.1 2833.83     357 2832.94
   378.1 2835.29   412.7 2845.36   436.2 2844.87   451.5 2846.34   464.2 2846.58
#Mann= 4 ,-1,0
       0      .1       0   220.3    .045       0   244.1      .1       0
  354.87     .06       0
#XS Ineff= 2 , 0
          178.74  2849.7
Permanent Ineff=
       F       F
Bank Sta=220.3,244.1
XS Rating Curve= 0 ,0
Exp/Cntr(USF)=0,0
Exp/Cntr=0.3,0.1

Type RM Length L Ch R = 1 ,26903   ,272.1,278.6,286.3
XS GIS Cut Line= 3
2162103.76463992425178.6247323362161643.93362569425197.017972906
2161548.51869023425170.577689587
#Sta/Elev= 30
       0 2892.75    17.8  2884.9    42.8 2869.77    59.6 2855.98    71.6 2847.42
    83.7 2837.16    94.4 2826.79   111.7 2816.06   123.7 2812.12   144.5  2811.9
   167.9 2811.01   176.2 2811.77   183.7  2813.9   199.7 2810.75   207.8 2812.36
   227.8 2814.07   303.8 2811.21   309.7 2814.36   319.8 2823.24   323.8 2825.68
   327.9 2826.55   351.9 2825.31   379.9 2825.33   395.9 2830.67   407.9 2832.65
   439.9 2832.64   468.2 2835.87   501.5 2845.59   538.8 2847.16   559.2  2853.5
#Mann= 7 ,-1,0
       0      .1       0      50     .08       0   144.5    .045       0
   176.2     .08       0     250      .1       0     350     .06       0
   550.2      .1       0
#XS Ineff= 2 , 0
                          230.14         2833.64
Permanent Ineff=
       F       F
Bank Sta=144.5,176.2
XS Rating Curve= 0 ,0
Exp/Cntr(USF)=0,0
Exp/Cntr=0.3,0.1

Type RM Length L Ch R = 1 ,26625   ,280.1,274.6,262.8
XS GIS Cut Line= 3
2162111.81168267425061.3678237072162017.54632475425045.273738209
 2161683.0192619 424829.15316152
#Sta/Elev= 30
       0 2864.82     7.7 2862.43      24 2854.56    80.8 2820.46      93 2815.34
   125.6 2812.72   140.1 2812.84   157.4 2810.74   168.7 2810.35   187.7 2806.71
   206.8 2804.65   221.1 2804.22   229.8  2802.4   240.1 2798.71   255.8 2800.15
   261.4 2799.48   268.7 2798.43   284.7 2799.21   299.2 2799.64   306.8 2801.26
   319.5  2802.2   335.4 2813.72   354.4 2818.46   373.5 2820.79   390.7 2818.59
   403.4 2821.04   435.4 2831.23   454.4 2840.44     483 2851.06   493.9  2853.8
#Mann= 5 ,-1,0
       0      .1       0   261.4    .045       0   284.7      .1       0
  285.63     .06       0  345.63      .1       0
Bank Sta=261.4,284.7
XS Rating Curve= 0 ,0
Exp/Cntr(USF)=0,0
Exp/Cntr=0.3,0.1

Type RM Length L Ch R = 1 ,26350   ,468.3,474.5,490.1
XS GIS Cut Line= 3
2162187.68380002424778.5717499542162053.18322835424718.793718104
2161724.40405318424692.353434785
#Sta/Elev= 30
       0 2836.52    38.9 2830.28    82.6 2819.71   115.8  2814.2   121.9 2811.02
   130.8 2803.56   140.1 2799.47   148.2  2794.4   153.3 2792.88   164.5 2791.13
   188.3 2791.01   201.6 2789.19   229.4 2789.09   252.5    2788   257.3 2789.11
   260.6 2791.62   268.6 2802.98   272.6  2806.6   276.6 2807.14   284.6 2807.38
   300.7 2805.38   324.8    2806   336.8 2804.55   387.3 2804.24   405.9 2807.45
   425.1 2814.54   441.1 2823.69   454.2 2833.01   473.2 2848.95     477 2850.83
#Mann= 5 ,-1,0
       0     .12       0      40      .1       0   229.4    .045       0
   257.3     .06       0  347.19      .1       0
Bank Sta=229.4,257.3
XS Rating Curve= 0 ,0
Exp/Cntr(USF)=0,0
Exp/Cntr=0.3,0.1

Type RM Length L Ch R = 1 ,25876   ,397.3,392.5,390.8
XS GIS Cut Line= 2
2162480.82607159424590.0410341192162053.18322835 424246.31735098
#Sta/Elev= 30
       0 2845.94    33.3 2842.92    88.1 2836.06   103.5 2834.88   108.6 2832.71
   116.3 2827.34   129.1 2817.07   139.4 2809.77   148.2 2802.45   165.1 2791.26
   180.3 2778.32   186.5 2777.38     201 2776.46   214.5 2777.62   251.4 2782.59
   274.2 2781.98   293.4 2782.25   307.8 2785.61   314.2 2786.26   339.8 2786.72
     351 2786.02   373.8 2786.91   382.3 2788.83   405.1 2796.22   433.5 2797.32
   459.1 2802.12     473 2806.03   503.8 2818.33     516 2821.47   548.7 2833.12
#Mann= 5 ,-1,0
       0      .1       0   186.5    .045       0   214.5      .1       0
     270     .06       0     430      .1       0
Bank Sta=186.5,214.5
XS Rating Curve= 0 ,0
Exp/Cntr(USF)=0,0
Exp/Cntr=0.3,0.1

Type RM Length L Ch R = 1 ,25483   ,374.4,375.4,375.5
XS GIS Cut Line= 3
2162715.33988885424293.4500299382162649.81396932424208.381292305
 2162280.7995804423998.008603294
#Sta/Elev= 30
       0 2841.51    42.4 2826.49    57.6 2819.33      97 2809.37   109.3 2802.42
   136.9 2780.89   141.5  2778.1   150.7 2775.29   162.3 2769.09   182.9 2768.58
   192.1 2769.04   204.8 2770.29   225.3 2770.69     235 2771.82     252 2771.43
   288.8 2773.36   310.3 2776.69   325.7 2775.66   348.1 2775.49     369 2776.23
   380.9 2777.96   396.5 2778.88   412.7 2781.91   428.8 2787.71   436.4 2789.56
   451.1 2790.78   465.8 2789.03   477.5  2790.1   495.1  2796.4   532.1  2814.6
#Mann= 5 ,-1,0
       0      .1       0   162.3    .045       0   192.1      .1       0
  277.38     .06       0  457.38      .1       0
Bank Sta=162.3,192.1
XS Rating Curve= 0 ,0
Exp/Cntr(USF)=0,0
Exp/Cntr=0.3,0.1

Type RM Length L Ch R = 1 ,25108   ,202.7,215.6,226.9
XS GIS Cut Line= 3
2163070.55934734424054.3379025382162979.74272203423971.568319976
2162637.16861643423765.793941107
#Sta/Elev= 30
       0 2841.45     8.6 2836.72    19.5 2832.34    35.7 2822.56    49.2 2815.83
    90.3 2790.41   102.7 2779.71   112.9 2766.23   116.9 2762.31   130.1 2755.35
   138.9 2754.26     203 2760.43   220.4 2759.72   228.5 2761.15   243.8 2762.16
   262.4 2758.69   267.3 2758.67   282.9 2762.85   290.4 2763.26   327.7 2761.12
   331.3 2759.08     337 2757.97   357.5 2758.99   377.9 2760.31   404.2  2763.4
     435 2765.22     445 2767.97   456.6 2774.74   500.4    2803   522.5 2818.17
#Mann= 5 ,-1,0
       0      .1       0   331.3    .045       0   357.5      .1       0
  402.88     .06       0  512.88      .1       0
#XS Ineff= 2 , 0
          287.72 2773.54
Permanent Ineff=
       F       F
Bank Sta=331.3,357.5
XS Rating Curve= 0 ,0
Exp/Cntr(USF)=0,0
Exp/Cntr=0.3,0.1

Type RM Length L Ch R = 1 ,24892   ,302.8,298.6,285
XS GIS Cut Line= 3
2163196.91775001423915.7454403712162966.91448748423779.810385873
2162911.73654901423627.572757962
#Sta/Elev= 30
       0 2833.91    20.8 2825.41    40.3 2814.94      55 2803.94    75.2 2787.26
    87.1 2780.23   121.7  2757.4   126.3 2751.95   130.8 2748.43   135.6 2748.06
   168.1 2749.73   191.4 2754.32   214.6 2751.76   251.8 2753.09   261.1 2756.02
   274.2  2757.2   278.5 2755.96   283.9 2752.93   302.42753.736     3262753.804
   333.8 2754.93     338 2758.16   342.3 2760.12   361.9 2759.92   367.8 2760.88
   372.1 2762.79   380.4 2769.82   406.1 2785.95   423.1 2800.55   429.1 2804.49
#Mann= 4 ,-1,0
       0      .1       0   302.4    .045       0     326     .06       0
  427.17      .1       0
#XS Ineff= 2 , 0
          266.67 2777.82
Permanent Ineff=
       F       F
Bank Sta=302.4,326
XS Rating Curve= 0 ,0
Exp/Cntr(USF)=0,0
Exp/Cntr=0.3,0.1

Type RM Length L Ch R = 1 ,24593   ,428.3,443.3,452.9
XS GIS Cut Line= 2
2163346.45889979423775.4057557532163095.87090811423516.433779218
#Sta/Elev= 30
       0  2812.6    25.4 2799.56    34.3 2795.61    47.6    2788    64.3 2780.36
    75.5 2773.67    89.6 2763.44     120 2746.97   124.8 2745.67   133.3 2744.86
   142.2 2745.46   152.8 2743.87   157.42742.564   164.4 2741.16   187.82742.369
   201.2  2742.8   220.2  2742.7   231.3 2743.71   239.1  2743.6   249.3 2745.09
   264.7 2744.96   274.8 2746.55   281.4 2748.28     287 2751.95   296.6 2760.25
   303.7 2765.65   331.5 2791.41   341.4 2798.25   348.4 2801.87   360.4 2803.98
#Mann= 5 ,-1,0
       0      .1       0   157.4    .045       0   187.8      .1       0
   201.2     .06       0   341.4      .1       0
#XS Ineff= 2 , 0
                           252.1         2750.29
Permanent Ineff=
       F       F
Bank Sta=157.4,187.8
XS Rating Curve= 0 ,0
Exp/Cntr(USF)=0,0
Exp/Cntr=0.3,0.1

Type RM Length L Ch R = 1 ,24150   ,359.9,348.8,341
XS GIS Cut Line= 2
2163576.03230427 423643.209219812163388.69374292423122.351249985
#Sta/Elev= 30
       0 2817.19      14 2809.82    46.9 2795.37    57.4 2789.74    65.9 2787.39
    74.4 2782.04    82.8 2778.28   112.7 2759.87   125.4 2749.19   142.4 2739.07
   150.9 2737.28   173.4 2736.47   184.9 2734.89   198.4 2735.01   214.7 2736.64
   245.3 2735.61   255.9 2733.51   265.7 2732.12   295.4 2732.53     304 2733.51
   316.7 2735.72   370.4 2734.17   393.2 2737.75   397.5 2740.16   404.8 2745.87
   413.2  2750.2   452.7 2765.61     474 2772.88   519.6  2797.5   553.5 2812.08
#Mann= 5 ,-1,0
       0      .1       0   255.9    .045       0     304      .1       0
     330     .06       0     430      .1       0
#XS Ineff= 2 , 0
          213.16 2749.99  334.77         2750.77
Permanent Ineff=
       F       F
Bank Sta=255.9,304
XS Rating Curve= 0 ,0
Exp/Cntr(USF)=0,0
Exp/Cntr=0.3,0.1

Type RM Length L Ch R = 1 ,23801   ,417.3,405.2,386.1
XS GIS Cut Line= 3
2163929.89164104423401.0698496112163834.09351308423310.380955137
2163602.90069759422954.011919108
#Sta/Elev= 30
       0 2803.33    75.5 2765.16    94.5 2753.13   104.6 2749.96   123.5 2739.27
   138.1 2732.46     162 2730.35   176.3 2724.47   185.8 2722.93   190.6  2723.5
   200.7  2726.6   216.3 2727.38     253 2726.02   290.7    2727   324.1 2724.51
   333.6 2722.87   351.1 2723.49   355.9 2724.62   365.5 2729.43   385.3 2731.47
   391.6    2734   400.4 2738.52   414.7 2747.89   438.5 2756.13   462.3 2771.15
   476.6 2778.05   495.7 2789.33   519.6 2797.55   547.7 2808.79   556.7 2811.43
#Mann= 3 ,-1,0
       0      .1       0   324.1    .045       0   355.9      .1       0
Bank Sta=324.1,355.9
XS Rating Curve= 0 ,0
Exp/Cntr(USF)=0,0
Exp/Cntr=0.3,0.1

Type RM Length L Ch R = 1 ,23396   ,447.1,455.3,465.6
XS GIS Cut Line= 3
2164166.19369002423116.2300824622164095.94172952422922.079209786
2163794.49695352422855.659174397
#Sta/Elev= 30
       0  2760.3     7.5 2758.11    28.8 2757.24      50 2752.39    96.8 2732.02
   113.8 2727.77   135.1 2725.97   152.1 2722.49   170.5 2724.15   185.1  2721.7
   222.6 2720.14   234.9 2717.67   275.9 2712.92   287.6 2713.21   304.4 2711.94
   317.8 2713.49     325 2714.77   340.8  2715.3   368.1 2719.46   374.8 2724.08
   390.5 2730.76   411.8 2737.43   427.4 2743.75   445.3 2755.44   448.7  2757.2
   456.1 2758.78   476.6  2771.7   488.7 2774.94     497  2779.7   515.1 2786.88
#Mann= 5 ,-1,0
       0      .1       0     190     .06       0   287.6    .045       0
   317.8     .06       0  386.47      .1       0
Bank Sta=287.6,317.8
XS Rating Curve= 0 ,0
Exp/Cntr(USF)=0,0
Exp/Cntr=0.3,0.1

Type RM Length L Ch R = 1 ,22941   ,272.4,273,273.5
XS GIS Cut Line= 2
 2164480.9224731422724.862797015  2164090.066111422394.934044304
#Sta/Elev= 30
       0 2778.26    63.8 2749.62      90 2739.57   105.3 2734.47   121.4 2733.31
   168.5    2721   184.2 2715.17   201.8 2711.15   215.6  2703.7   224.5  2702.3
     229 2702.09   257.5 2702.26   267.1 2703.29   275.6 2707.86   278.4 2708.47
     287 2707.81   298.4 2709.23   340.9  2706.9   349.4 2708.91   362.2  2716.2
   383.5 2734.13   398.8  2743.8   409.1  2748.5   421.2 2758.79   430.2 2765.14
   440.3 2770.52   460.1 2783.64   472.1 2788.89   485.7 2797.54   511.5 2815.63
#Mann= 5 ,-1,0
       0      .1       0     220     .06       0   224.5    .045       0
   257.5     .06       0     340      .1       0
Bank Sta=224.5,257.5
XS Rating Curve= 0 ,0
Exp/Cntr(USF)=0,0
Exp/Cntr=0.3,0.1

Type RM Length L Ch R = 1 ,22668   ,223.5,220.6,216.8
XS GIS Cut Line= 2
2164623.10258086 422495.445197682164329.33157953422235.842530351
#Sta/Elev= 30
       0 2733.56     9.5 2730.25    26.4 2725.15    46.2 2720.13    75.9 2708.74
      82 2707.26   100.1 2704.84     132 2702.59   196.1 2701.35   199.2 2700.28
   202.8  2697.5   204.9    2696   207.7 2695.23   221.9 2694.55     233 2694.85
   237.1 2697.79     239 2699.48   244.1 2700.85   263.2 2700.08   265.5 2700.38
   267.2 2701.24   272.9 2705.72     283  2712.8   302.8 2730.84   317.5  2741.8
   324.2 2745.75   340.2 2751.17   347.7 2752.65   377.9 2755.82     392 2756.57
#Mann= 5 ,-1,0
       0     .12       0      20      .1       0   202.8    .045       0
   237.1     .06       0     360      .1       0
#XS Ineff= 2 , 0
                          244.76         2707.85
Permanent Ineff=
       F       F
Bank Sta=202.8,237.1
XS Rating Curve= 0 ,0
Exp/Cntr(USF)=0,0
Exp/Cntr=0.3,0.1

Type RM Length L Ch R = 1 ,22447   ,356.3,346.3,334.4
XS GIS Cut Line= 2
2164866.03094752422366.194605914 2164448.7343021422078.800222019
#Sta/Elev= 30
       0 2791.76    22.2 2779.21      51 2759.36    60.5 2756.84    65.3 2753.98
    79.7 2740.14    89.7 2733.25    94.5 2728.37   114.2 2712.86   128.5 2702.73
   137.2 2698.67   156.9  2696.3   199.3 2697.24   213.4 2695.81   246.5 2696.03
   264.5 2698.38   278.2 2698.61     284 2697.42   293.7 2692.81   303.4 2691.44
   327.7 2691.52   337.4 2692.82   351.9 2697.46   376.2 2696.76   387.5 2697.82
   405.4 2702.42   417.9    2710   433.5 2716.88   473.7  2745.6   506.7 2767.58
#Mann= 5 ,-1,0
       0     .12       0      20      .1       0   293.7    .045       0
   337.4     .06       0     430      .1       0
Bank Sta=293.7,337.4
XS Rating Curve= 0 ,0
Exp/Cntr(USF)=0,0
Exp/Cntr=0.3,0.1

Type RM Length L Ch R = 1 ,22101   ,405.3,404.9,402.3
XS GIS Cut Line= 2
2165081.00194667421937.402185143 2164516.5593767421830.491474334
#Sta/Elev= 30
       0 2792.32      66 2765.19    86.3 2754.19    94.5 2748.53   106.2 2737.27
   110.8 2731.99   118.9 2718.93     123  2713.8   147.4  2696.4   161.8 2688.15
   188.1 2685.44     220 2688.14   253.3 2686.82     309 2688.94   314.3 2688.46
   322.2  2684.7     351 2683.12   363.7 2684.96   375.4 2688.02   403.9 2685.44
     408 2686.37   416.1 2690.75   428.3 2702.65   432.4 2704.31   444.6 2704.85
   448.7 2706.33   452.7 2709.75   476.7 2721.07   533.1 2754.41   574.5 2773.67
#Mann= 5 ,-1,0
       0      .1       0   322.2    .045       0   363.7      .1       0
     380     .06       0  574.48      .1       0
#XS Ineff= 2 , 0
          309.57 2703.39
Permanent Ineff=
       F       F
Bank Sta=322.2,363.7
XS Rating Curve= 0 ,0
Exp/Cntr(USF)=0,0
Exp/Cntr=0.3,0.1

Type RM Length L Ch R = 1 ,21696   ,368,374.4,374
XS GIS Cut Line= 2
2165129.28420317421547.6954005812164567.14078827421443.083844843
#Sta/Elev= 30
       0 2760.48    21.5 2749.28    41.8 2733.52    66.2 2710.19    90.6 2689.48
    98.8 2683.22   106.9 2679.47   140.3 2678.01   200.5 2679.88     229 2679.11
   241.2 2676.93     290 2677.96   298.2 2679.06   330.7 2678.42     347 2675.97
   359.2 2677.12   375.4 2676.99   383.6 2675.12   399.9 2675.03   405.42676.623
   412.1 2680.77   444.6 2680.92   452.8 2686.44     465 2696.58   481.2 2712.16
   493.1 2719.64     526 2735.15   538.2 2739.29   550.4 2744.95   571.8 2749.74
#Mann= 5 ,-1,0
       0      .1       0     330     .06       0   375.4    .045       0
   405.4     .06       0     430      .1       0
#XS Ineff= 2 , 0
          226.09 2701.48
Permanent Ineff=
       F       F
Bank Sta=375.4,405.4
XS Rating Curve= 0 ,0
Exp/Cntr(USF)=0,0
Exp/Cntr=0.3,0.1

Type RM Length L Ch R = 1 ,21322   ,366.4,369.7,379.6
XS GIS Cut Line= 3
  2165150.085314421341.052441139  2164946.129637421184.473936696
2164610.82473462421048.778750139
#Sta/Elev= 30
       0 2754.64    49.8 2726.08    65.5 2713.05    78.1 2700.32   112.5 2674.99
   118.4 2672.61   149.6 2672.14   163.8 2670.67   183.9 2672.47   199.1  2670.8
   224.3 2670.46   239.4 2668.18   254.5 2671.69     274 2667.12   280.8 2665.33
   293.8 2664.92   311.72666.939   319.6 2671.34     324 2672.08     393 2673.61
   427.5 2673.03   444.8  2675.4   479.3 2694.15   500.9 2701.78   513.8 2708.55
   526.8 2711.44   543.1 2721.26   569.9    2733   595.8 2746.94   618.8 2756.47
#Mann= 4 ,-1,0
       0      .1       0     274    .045       0   311.7     .06       0
  407.13      .1       0
#XS Ineff= 2 , 0
          259.03 2688.77
Permanent Ineff=
       F       F
Bank Sta=274,311.7
XS Rating Curve= 0 ,0
Exp/Cntr(USF)=0,0
Exp/Cntr=0.3,0.1

Type RM Length L Ch R = 1 ,20952   ,397.9,399.3,397.7
XS GIS Cut Line= 3
2165364.90762975421073.696756768 2164909.3343101420701.858097111
2164835.53427078420538.646471689
#Sta/Elev= 30
       0 2791.75    45.1 2766.02    57.7  2760.9    77.6 2747.93    93.9 2740.35
   119.7 2724.18   171.5 2696.87     180 2690.45   199.9 2667.94   205.6 2662.61
   209.6 2660.09   217.8 2658.58   233.3 2658.29   251.1 2659.85   264.3 2663.26
   285.5 2664.25   323.4 2665.14   398.5 2662.13   424.7 2665.32   506.9 2664.25
   538.5 2665.63   582.8 2669.47   588.8 2671.58   593.2  2674.4   615.1 2692.12
   628.7 2701.83   654.7 2713.06   685.4 2729.83   724.9 2748.63   767.2 2766.52
#Mann= 4 ,-1,0
       0      .1       0   209.6    .045       0   251.1     .06       0
     340      .1       0
#XS Ineff= 2 , 0
                           282.9         2690.49
Permanent Ineff=
       F       F
Bank Sta=209.6,251.1
XS Rating Curve= 0 ,0
Exp/Cntr(USF)=0,0
Exp/Cntr=0.3,0.1

Type RM Length L Ch R = 1 ,20553   ,601.9,640.9,679
XS GIS Cut Line= 2
2165617.42571301420766.3367639452165081.27158119420354.584407808
#Sta/Elev= 30
       0  2747.6    81.6 2706.45   107.5 2691.65   126.7 2683.15   161.5 2660.05
   167.2 2656.65   172.6 2654.47   184.3  2653.1   225.2    2653   268.9 2654.13
   284.3 2652.04   297.4 2650.73   324.4 2650.57   332.6 2651.89   339.5 2654.27
   359.7 2654.01   366.9 2654.94   415.1 2657.12   478.1 2655.11   500.9 2655.74
   507.6 2659.74   523.8 2671.46   540.9 2685.41   546.6 2687.67   551.3  2690.5
   571.5 2705.87     615 2729.56     627 2734.93   657.2 2750.93     676 2762.41
#Mann= 5 ,-1,0
       0      .1       0     280     .06       0   284.3    .045       0
   332.6     .06       0     470      .1       0
#XS Ineff= 2 , 0
          265.12 2666.96  349.19            2665
Permanent Ineff=
       F       F
Bank Sta=284.3,332.6
XS Rating Curve= 0 ,0
Exp/Cntr(USF)=0,0
Exp/Cntr=0.3,0.1

Type RM Length L Ch R = 1 ,19912   ,499.2,471,429.6
XS GIS Cut Line= 4
 2165839.9471991420652.4478143752165756.37023149420488.447726994
2165951.90879721 420195.139878412165865.17798177420106.832139052
#Sta/Elev= 30
       0 2760.97    21.6 2749.27    46.9 2733.29    53.1 2730.66    75.5 2717.18
    84.5 2712.97    97.9 2703.38   124.2  2688.9   142.8  2672.3     151 2668.39
   174.7 2652.06   183.2 2648.37   197.6 2645.31   207.2 2644.62   255.5 2643.06
   284.4 2643.67   322.6  2642.6   351.4 2643.32   365.1 2641.34   385.1 2641.09
   409.1 2639.98   421.7 2640.22     424 2641.06   428.9 2643.53   495.7 2645.81
   529.3 2654.32   574.5 2654.33   584.2 2657.02   625.5 2658.26   660.4 2661.56
#Mann= 5 ,-1,0
       0      .1       0   385.1    .045       0     424      .1       0
  424.07     .06       0  546.58      .1       0
#XS Ineff= 2 , 0
                          458.76         2660.79
Permanent Ineff=
       F       F
Bank Sta=385.1,424
XS Rating Curve= 0 ,0
Exp/Cntr(USF)=0,0
Exp/Cntr=0.3,0.1

Type RM Length L Ch R = 1 ,19441   ,448.8,442.4,438.1
XS GIS Cut Line= 3
2166437.60136368420456.9092486522166368.21671133 420299.21685694
2165970.83188422419969.639758262
#Sta/Elev= 30
       0 2782.93    43.4 2758.14    56.5  2749.2    87.1 2722.16   104.6 2705.25
   113.3 2699.38   161.7 2658.23   172.3 2649.99   182.7 2643.41   190.8 2640.24
   206.8 2640.68   219.1 2639.31   231.9 2635.07   247.6 2633.74   260.7 2629.96
   273.2 2630.15   293.1 2629.48   301.6 2629.97   319.6 2635.15   325.9 2635.89
   349.9 2635.33   385.4 2637.05   501.3 2636.11   511.8 2639.52   531.7  2652.8
   541.3  2655.6   560.1 2654.89   572.5 2657.29   645.3 2659.72   688.6  2662.5
#Mann= 5 ,-1,0
       0      .1       0   273.2    .045       0   301.6      .1       0
  412.28     .06       0  532.28      .1       0
#XS Ineff= 2 , 0
                           328.7          2672.2
Permanent Ineff=
       F       F
Bank Sta=273.2,301.6
XS Rating Curve= 0 ,0
Exp/Cntr(USF)=0,0
Exp/Cntr=0.3,0.1

Type RM Length L Ch R = 1 ,18999   ,523,506,482.4
XS GIS Cut Line= 2
2166779.16438201420014.2219282652166198.85638051 419672.02943825
#Sta/Elev= 30
       0 2718.19    20.5 2707.32    32.2 2703.12    43.8 2695.35   120.2 2650.28
   138.1  2638.5   157.8 2628.54   161.4 2627.32   184.6 2626.19   207.8  2627.5
   216.2 2625.65   222.6 2623.34   249.6 2623.09   261.9 2623.39   269.8 2625.74
   277.5 2627.94   300.9 2627.02   328.5 2628.57   359.3 2625.91   411.9 2626.84
     440 2625.59   464.5 2626.44   474.5 2628.36   495.7 2641.87     505 2644.53
   528.2 2642.83   537.5 2645.53   561.2 2646.43   616.6 2652.93   673.7 2656.82
#Mann= 5 ,-1,0
       0      .1       0   216.2    .045       0   269.8      .1       0
     460     .06       0     630      .1       0
#XS Ineff= 2 , 0
                          279.32         2649.47
Permanent Ineff=
       F       F
Bank Sta=216.2,269.8
XS Rating Curve= 0 ,0
Exp/Cntr(USF)=0,0
Exp/Cntr=0.3,0.1

Type RM Length L Ch R = 1 ,18493   ,383.4,400.7,417.7
XS GIS Cut Line= 2
 2167017.2798935419397.6446766712166184.66406526419591.606318477
#Sta/Elev= 30
       0 2732.75     9.3 2725.39    17.6 2723.48    30.5 2714.67    62.7 2697.41
    95.6 2682.83   147.1 2656.49   170.4  2648.1   202.4 2639.41   233.7 2615.45
   239.3 2613.32   255.8 2613.03   276.3 2615.17   283.7 2617.86   313.3 2619.14
   333.6 2617.66   370.8 2618.01   387.2 2619.65   469.3 2617.65   510.2 2618.33
   564.3 2621.49   584.3 2621.11   600.8 2624.19   621.3 2624.85   629.5 2626.89
   641.8  2632.4     650 2633.68   695.2 2637.94   744.5 2649.69   854.9 2658.51
#Mann= 7 ,-1,0
       0      .1       0   233.7    .045       0   276.3      .1       0
     450     .06       0     460      .1       0     550     .06       0
     650      .1       0
#XS Ineff= 2 , 0
                          387.44          2644.5
Permanent Ineff=
       F       F
Bank Sta=233.7,276.3
XS Rating Curve= 0 ,0
Exp/Cntr(USF)=0,0
Exp/Cntr=0.3,0.1

Type RM Length L Ch R = 1 ,18092   ,445.8,443.7,440.5
XS GIS Cut Line= 3
2167036.63128083  419141.05384672166888.67298737419119.638830542
2166265.69069912418872.392734895
#Sta/Elev= 30
       0 2719.95     8.5 2717.29    24.7 2705.89   117.7 2653.87   154.3 2621.79
   171.6 2610.94   176.4 2609.31   193.1  2608.8     206 2606.86   244.7 2609.11
   266.2 2606.93   283.4 2605.49   309.3 2605.58   315.1 2607.18   322.2 2611.04
     391 2610.27   412.5 2607.31     447  2609.6   469.1 2607.53   524.4 2611.44
   584.7 2610.42   644.7 2611.39   650.9 2614.42   696.6 2647.62   700.9 2649.76
   718.1 2655.68     731 2662.43   739.6 2663.47   765.4 2673.01   819.8 2689.08
#Mann= 5 ,-1,0
       0      .1       0   266.2    .045       0   315.1      .1       0
   379.5     .06       0   479.5      .1       0
#XS Ineff= 2 , 0
                          332.37         2623.67
Permanent Ineff=
       F       F
Bank Sta=266.2,315.1
XS Rating Curve= 0 ,0
Exp/Cntr(USF)=0,0
Exp/Cntr=0.3,0.1

Type RM Length L Ch R = 1 ,17648   ,441.9,443.7,445.7
XS GIS Cut Line= 2
2167106.71678825418736.1153593412166384.44669782418492.762902996
#Sta/Elev= 30
       0 2686.61      58 2656.03   108.2 2633.56   116.6 2628.54   125.1 2626.87
   146.2 2617.96   192.6 2601.47   212.7  2597.8   230.6 2597.13   247.2  2595.5
   259.8 2597.34   269.5 2601.28   307.4  2600.1   332.7  2600.9     353 2599.07
   383.2 2602.91   417.9 2602.04   446.3 2604.43   479.6  2603.4   500.8 2604.55
   517.6 2603.49   593.6 2603.83   602.1  2606.5   618.9 2614.71   631.6 2623.77
   645.2 2631.56   669.6 2640.48   705.2 2658.45   724.5 2664.76   762.2 2685.52
#Mann= 5 ,-1,0
       0      .1       0     140     .06       0   230.6    .045       0
   259.8     .06       0     350      .1       0
#XS Ineff= 2 , 0
                          285.22         2617.03
Permanent Ineff=
       F       F
Bank Sta=230.6,259.8
XS Rating Curve= 0 ,0
Exp/Cntr(USF)=0,0
Exp/Cntr=0.3,0.1

Type RM Length L Ch R = 1 ,17205   ,467.3,465,462.2
XS GIS Cut Line= 2
2167295.23096429418405.5442073392166636.07676694418005.005532391
#Sta/Elev= 30
       0 2680.27      52  2650.6    69.1 2638.31      84 2632.71    97.2 2621.86
   113.1 2606.12   115.9 2602.81   121.9    2591   125.3 2589.06   139.3 2588.69
   162.6 2588.75   174.3 2590.79   214.2 2592.76   229.6 2591.22   244.1  2593.1
   316.9 2594.74   359.3 2593.31   415.5 2595.05   448.2 2593.21   503.3  2595.4
   546.9 2593.84   578.4 2595.68   613.9 2594.93   628.4  2597.8   654.2 2609.37
   682.3 2613.16     700 2617.97   719.7 2626.59   740.2 2632.69   771.3 2651.37
#Mann= 6 ,-1,0
       0      .1       0   121.9    .045       0   174.3     .06       0
     360      .1       0     380     .07       0     610      .1       0
#XS Ineff= 2 , 0
                          246.02         2615.82
Permanent Ineff=
       F       F
Bank Sta=121.9,174.3
XS Rating Curve= 0 ,0
Exp/Cntr(USF)=0,0
Exp/Cntr=0.3,0.1

Type RM Length L Ch R = 1 ,16740   ,425.6,431.5,436.1
XS GIS Cut Line= 3
  2167628.243886418130.0522654712167556.85587798 418014.78049471
2166846.96034421417671.632416682
#Sta/Elev= 30
       0  2638.4    15.1 2635.48    23.9 2631.75    68.5 2618.65    99.8 2604.15
   128.1 2589.46   155.3 2584.94   176.3 2583.62   216.3 2584.68   226.8  2582.3
   245.1  2580.3   265.2 2580.72   275.1  2582.3     283 2584.09   318.5  2587.3
   367.4 2584.46   380.7 2587.34   527.3 2585.27   550.6 2588.68   628.5 2586.62
   681.5 2589.03   793.2 2591.34   798.3 2592.77   819.4 2603.95   838.8 2610.33
   856.1 2620.25     865 2623.35   878.3 2631.43     898 2641.26   924.1 2652.37
#Mann= 7 ,-1,0
       0      .1       0   226.8    .045       0   275.1     .06       0
  345.59     .05       0  565.59      .1       0  675.59     .07       0
  785.59      .1       0
#XS Ineff= 2 , 0
                          317.87         2604.87
Permanent Ineff=
       F       F
Bank Sta=226.8,275.1
XS Rating Curve= 0 ,0
Exp/Cntr(USF)=0,0
Exp/Cntr=0.3,0.1

Type RM Length L Ch R = 1 ,16308   ,438.4,443,445.9
XS GIS Cut Line= 3
2168055.54276457417955.2778198752167934.40731964417797.369114868
2167233.55224536417271.727809162
#Sta/Elev= 30
       0 2688.85    43.8 2666.76    73.2 2653.26    83.3 2646.76    93.4  2644.7
   128.7 2626.68   184.1 2591.56     206 2580.27   212.7 2577.96   360.8 2577.49
   379.3 2575.25   446.5 2577.54     515 2578.09     535 2575.44   546.5 2573.53
   561.8 2573.38   572.7 2573.48   579.12575.503   586.8 2579.65   609.2 2577.27
   671.8 2578.18   686.5 2577.43   716.8 2579.53   781.8 2578.46     946 2582.12
   952.2 2584.62     986  2603.5   999.3 2609.57  1026.5 2619.35  1075.1 2640.64
#Mann= 5 ,-1,0
       0      .1       0     535    .045       0   579.1     .06       0
  659.02     .07       0  909.02      .1       0
#XS Ineff= 2 , 0
                          589.06          2589.4
Permanent Ineff=
       F       F
Bank Sta=535,579.1
XS Rating Curve= 0 ,0
Exp/Cntr(USF)=0,0
Exp/Cntr=0.3,0.1

Type RM Length L Ch R = 1 ,15865   ,510.3,500.2,489.6
XS GIS Cut Line= 2
2168377.84957342417702.1912652752167696.46269566417005.662456891
#Sta/Elev= 30
       0 2647.34      33 2632.42    44.3 2630.05    53.9 2625.33    75.4 2617.36
   122.5 2601.51   137.7 2591.51   156.8 2575.13     166 2570.86     242  2569.5
   264.4 2570.73   294.1 2570.45   322.7 2568.77   404.3 2569.97   426.2 2568.14
     446  2569.6   517.2 2571.17   528.6 2571.09   536.5 2569.19   576.1 2568.55
   587.4 2569.44   595.9 2571.15   654.5 2571.55   677.9 2580.43   697.7 2581.31
     709 2587.49     740 2590.33   768.5 2590.46     796 2593.47   974.4  2604.6
#Mann= 8 ,-1,0
       0      .1       0     520     .06       0   536.5    .045       0
   587.4     .06       0     600     .08       0     650      .1       0
     740     .07       0     790      .1       0
Bank Sta=536.5,587.4
XS Rating Curve= 0 ,0
Exp/Cntr(USF)=0,0
Exp/Cntr=0.3,0.1

Type RM Length L Ch R = 1 ,15365   ,464.4,477.2,483.7
XS GIS Cut Line= 3
2168897.00148029 417327.969265742168468.70115713 416992.68365922
2167984.15937738416756.902168183
#Sta/Elev= 30
       0 2661.68    30.5 2649.73    45.3 2640.55    56.7 2637.81   108.4 2605.67
   136.5 2586.23   153.6 2568.24   158.5 2560.82   162.1 2559.06   204.9 2556.84
   239.8 2559.43   296.5 2555.83   326.2 2560.59   354.9 2558.81   453.2 2560.74
   510.7 2556.58   536.6 2560.66     629 2562.21   642.7 2559.74   655.7 2562.26
   693.6 2562.35   705.5 2560.57   731.3  2563.8     7772563.766   809.82563.998
   824.8 2564.79   851.5 2570.71   931.5 2569.59   949.3 2577.83  1082.8 2603.91
#Mann= 6 ,-1,0
       0      .1       0  673.93     .08       0     777    .045       0
   809.8     .08       0  883.93     .06       0 1003.93      .1       0
#XS Ineff= 2 , 0
          728.12 2607.24
Permanent Ineff=
       F       F
Bank Sta=777,809.8
XS Rating Curve= 0 ,0
Exp/Cntr(USF)=0,0
Exp/Cntr=0.3,0.1

Type RM Length L Ch R = 1 ,14888   ,502,498.7,494.3
XS GIS Cut Line= 3
2169039.76825468416966.7260638762168739.09277529416767.717832909
2168312.95558506416270.197255492
#Sta/Elev= 30
       0 2625.43    57.1 2590.94    81.1 2573.68     105 2553.65   114.6 2550.15
   124.2 2549.55   176.9 2553.31   220.2 2550.59   249.1 2555.35   286.6 2553.72
   306.5 2550.07   329.9  2553.8     353 2553.15   363.9 2555.12   412.7 2556.22
   432.4 2554.09   474.5 2556.64   590.4 2557.39   668.32554.052   691.62554.124
   740.1 2554.18   753.1 2552.29   790.5  2554.1     807 2551.41   822.1 2553.89
   860.9 2554.33   886.4 2565.57   909.1 2565.98   920.5 2569.23  1015.6 2583.15
#Mann= 6 ,-1,0
       0      .1       0  650.57     .08       0   668.3    .045       0
   691.6     .08       0  780.57     .06       0  910.57      .1       0
#XS Ineff= 2 , 0
          605.22  2587.1
Permanent Ineff=
       F       F
Bank Sta=668.3,691.6
XS Rating Curve= 0 ,0
Exp/Cntr(USF)=0,0
Exp/Cntr=0.3,0.1

Type RM Length L Ch R = 1 ,14389   ,387.8,392.7,403.7
XS GIS Cut Line= 2
2169292.85480928416614.1353937932168646.07805864416023.600099729
#Sta/Elev= 30
       0 2603.51     6.8 2600.12    15.3 2592.55    23.8 2589.19    44.3 2575.79
    78.5  2547.3    84.5 2545.18    98.4 2545.63   117.2 2543.09   130.9  2543.6
   142.7 2546.63   165.4 2546.07   174.2 2543.96     215 2543.95   228.4 2547.93
   345.5 2545.68   369.2 2547.34   454.2 2547.66   519.3 2544.11   561.8 2543.76
   671.8 2546.58     678 2544.85   688.8 2543.43   703.3 2545.02   754.8 2547.66
   770.1 2554.06   791.1 2554.49   805.3 2558.95   837.9 2562.21   875.8 2568.57
#Mann= 12 ,-1,0
       0      .1       0     210     .08       0     250      .1       0
     340     .08       0     390      .1       0     470     .08       0
     540      .1       0     610     .08       0     678    .045       0
   703.3      .1       0     740     .06       0     870      .1       0
#XS Ineff= 2 , 0
          452.17 2564.52
Permanent Ineff=
       F       F
Bank Sta=678,703.3
XS Rating Curve= 0 ,0
Exp/Cntr(USF)=0,0
Exp/Cntr=0.3,0.1

Type RM Length L Ch R = 1 ,13996   ,575.6,569.4,561.1
XS GIS Cut Line= 3
 2169513.4943697416356.7225733042169184.69816202416125.267348157
2168933.77474036415742.392816841
#Sta/Elev= 30
       0 2607.14      15 2597.12    26.1 2587.28    35.9  2584.5    60.9 2559.73
    70.1 2546.78    75.6 2542.78    84.8 2540.48   135.5 2542.22   149.9 2538.34
   195.8 2541.17     212 2540.12   226.6 2543.02   295.1 2541.16   339.1 2543.11
   378.3 2540.34   445.2 2542.07   558.5 2540.47   587.4 2542.52   607.8 2537.99
     622 2537.05   674.1  2540.9   713.1 2538.89   726.1 2536.54   756.1 2538.69
   769.4 2545.15   799.1 2554.29   827.2 2554.38   840.9 2559.96   859.9 2561.67
#Mann= 4 ,-1,0
       0      .1       0   713.1    .045       0   756.1     .06       0
  842.09     .12       0
#XS Ineff= 2 , 0
           591.3 2564.34
Permanent Ineff=
       F       F
Bank Sta=713.1,756.1
XS Rating Curve= 0 ,0
Exp/Cntr(USF)=0,0
Exp/Cntr=0.3,0.1
